--- LONGHOLLOW.prj (project) ---

Proj Title=LONGHOLLOW
Current Plan=p01
Default Exp/Contr=0,0
English Units
Geom File=g01
Flow File=f01
Plan File=p01
BEGIN DESCRIPTION:
END DESCRIPTION:
DSS Export Rating Curves= 0
DSS Export Rating Curve Sorted= 0
DSS Export Volume Flow Curves= 0
DXF OffsetX= 0
DXF OffsetY= 0
DXF ScaleX= 0
DXF ScaleY= 0

--- LONGHOLLOW.p01 (plan) ---

Plan Title=Floodplain
Program Version=4.00
Geom File=g01
Flow File=f01
K Sum by GR=0
Std Step Tol=0.01
Critical Tol=0.01
Num of Std Step Trials=20
Max Error Tol=0.3
Flow Tol Ratio=0.001
Split Flow NTrial=30
Split Flow Tol=0.02
Split Flow Ratio=0.02
Log Output Level=0
Friction Slope Method=1
Unsteady Friction Slope Method=2
Unsteady Bridges Friction Slope Method=1
Global Log Level=0
CheckData=False
Run HTab=0
Run UNet=0
Run PostProcess=0
UNET Theta=0
UNET Theta Warmup=0
UNET ZTol=0
UNET ZSATol=0
UNET MxIter=0
UNET MaxInSteps=0
UNET DtIC=0
UNET DtMin=0
UNET MaxCRTS=0
UNET WFStab=0
UNET SFStab=0
UNET WFX=0
UNET SFX=0
UNET DSS MLevel=0
UNET DZMax Abort=0
UNET Convert EG Bridges=0
UNET Use Existing IB Tables=0
UNET Froude Limit=0
UNET Froude Power=0
Write IC File=0
Echo Input=False
Echo Output=False
Write Detailed=0

--- LONGHOLLOW.f01 (steady flow) ---

Flow Title=NFF Regression Equation
Program Version=4.00
Number of Profiles=1
Profile Names=P100yr
River Rch & RM=LONGHOLLOW,Main      ,27474.8
530.7852
River Rch & RM=LONGHOLLOW,Main      ,26639.9
537.5564
River Rch & RM=LONGHOLLOW,Main      ,26282.6
631.1885
River Rch & RM=LONGHOLLOW,Main      ,24187.7
664.4534
River Rch & RM=LONGHOLLOW,Main      ,21819.8
734.4664
River Rch & RM=LONGHOLLOW,Main      ,21274.1
901.3978
River Rch & RM=LONGHOLLOW,Main      ,19969.1
929.8723
River Rch & RM=LONGHOLLOW,Main      ,15565.4
1014.589
River Rch & RM=LONGHOLLOW,Main      ,13683.9
1125.900
River Rch & RM=LONGHOLLOW,Main      ,13106.5
1181.563
River Rch & RM=LONGHOLLOW,Main      ,8780.7
1288.712
River Rch & RM=LONGHOLLOW,Main      ,5771.2
1423.165
River Rch & RM=LONGHOLLOW,Main      ,109.7
1539.892
Boundary for River Rch & Prof#=LONGHOLLOW,Main      ,1
Up Type=0
Dn Type=3
Dn Slope=0.003158

--- LONGHOLLOW.g01 (geometry) ---

Geom Title=USGS 10m DEM
Program Version=4.10

River Reach=LONGHOLLOW      ,Main
Reach XY= 30
     2294814.108      392835.889     2296038.093      392773.087
     2296317.088      393224.246     2296408.962      393836.488
     2297218.666      395124.673     2298726.998      394706.241
     2299013.295      396254.092     2299585.003      397534.708
     2299702.741      398262.873     2300363.513      398797.505
     2300463.139      399151.434     2300974.523      399753.411
     2301381.685      400785.763     2301600.818      400824.032
     2302392.716      402144.112      2302769.16      402429.525
     2302850.581      402881.591     2303230.137      403529.944
      2303578.96       403654.34     2303654.974      404120.992
     2304051.948        404571.3     2304199.809      405077.912
     2305504.304       406698.49     2305783.676      407623.712
     2306415.931      408662.122     2306372.421      408900.898
     2306648.436      409550.769     2307565.244      410043.662
     2307889.117      410806.385     2308579.943      411578.484

Type RM Length L Ch R = 1 ,27474.8 ,367.1,397.9,426.7
XS GIS Cut Line= 2
     2294921.865      393064.204     2294778.636      392699.621
#Sta/Elev= 30
       0  719.92       8  718.94      44  717.53   119.9  717.12  174.55715.3735
   199.8  715.19   219.8  714.55   231.8  714.97   239.8  713.83     244  712.01
   247.8  711.09   251.8  710.84   259.8  712.35   267.8  714.48   271.8  715.89
   275.8  717.88   279.8  720.68   287.8  727.31   291.8  732.08   295.8  737.58
   299.8  741.99   307.8  748.73   323.8  759.64   335.8  767.16   359.7   780.5
   363.7  782.18   371.7  783.99   379.7  787.47   383.7  788.71   391.7  790.38
#Mann= 4 ,-1 , 0
       0     .06       0  174.55     .12       0     244    .045       0
   259.8     .12       0
#XS Ineff= 2 , 0
          232.09  716.45
Permanent Ineff=
       F       F
Bank Sta=244,259.8
XS Rating Curve= 0 ,0
Exp/Cntr=0.3,0.1

Type RM Length L Ch R = 1 ,27076.9 ,43.6,47,57.2
XS GIS Cut Line= 4
     2295081.151      393053.413     2295120.344      392885.401
      2295293.13      392710.726     2295290.613      392677.892
#Sta/Elev= 30
       0  726.85     7.8  725.09   16.24722.0977    19.6  721.15    35.3  718.66
      98   712.6   121.6  710.98   141.2  710.36   152.9  709.58  178.15 709.275
   212.2  708.42   243.8  708.22   267.6  707.45   275.6  707.69   291.4  706.02
  292.68  705.49   299.3  704.05   303.3  704.21  308.73  705.71   315.2  706.88
   342.9  707.34  374.78707.3032   414.3  707.66   418.2  707.81   421.9  708.67
   425.5   711.1   432.8   718.3   440.2  724.57   443.8  727.18   451.2  731.42
#Mann= 6 ,-1 , 0
       0    .016       0   16.24     .06       0  178.15    .016       0
  292.68    .045       0  308.73    .016       0  374.78     .08       0
#XS Ineff= 2 , 0
          276.64  708.62  349.17          709.51
Permanent Ineff=
       F       F
Bank Sta=292.68,308.73
XS Rating Curve= 0 ,0
Exp/Cntr=0.3,0.1

Type RM Length L Ch R = 1 ,27029.9 ,174.2,148.7,114.9
XS GIS Cut Line= 5
     2295139.311      393056.017     2295155.804      392970.079
     2295200.335      392859.489      2295357.28      392734.836
     2295360.795      392712.245
#Sta/Elev= 30
       0   723.9       8  722.96    31.8  720.82    47.7  718.63    64.5 716.919
   99.62713.5208  101.15713.3869   111.4  712.62  152.49708.5801     159   707.9
     163   707.7   178.9  707.73   186.9  707.97  197.53707.8332  228.63707.5871
   230.3  707.57   234.2  706.63   241.3703.5923   242.1  703.26     246  703.07
   264.7  703.78   273.5  704.45  289.79704.7557   312.8   706.3  326.37706.2625
   356.1  705.59  374.45705.5847   403.2  705.69   418.6  707.07     430  707.22
#Mann= 12 ,-1 , 0
       0     .12       0    64.5    .016       0   99.62     .06       0
  101.15     .12       0  152.49     .06       0  197.53     .12       0
  228.63     .06       0   241.3    .045       0   264.7     .08       0
  289.79    .016       0  326.37     .06       0  374.45    .016       0
#XS Ineff= 2 , 0
                          329.27          708.13
Permanent Ineff=
       F       F
Bank Sta=241.3,264.7
XS Rating Curve= 0 ,0
Exp/Cntr=0.3,0.1

Type RM Length L Ch R = 1 ,26881.2 ,123.7,122.2,120.6
XS GIS Cut Line= 2
     2295406.978      393055.893     2295373.558      392718.479
#Sta/Elev= 30
       0  729.28      12  726.84    39.9  723.62    43.9  722.75    51.9   720.5
   59.35719.1077    71.8  717.53    79.8  715.88    99.7   713.9   119.7  711.16
   127.6  709.43   139.6  705.71   143.6  704.69   147.6  704.08   155.6  703.86
  188.88704.2924  231.46704.0413   243.3  703.92  250.26  701.99   251.3  701.32
   255.3  700.52   259.3  700.42   263.3  700.48   267.3  701.91   271.2  703.63
   275.2  704.19   287.2  704.45   307.2  704.12  321.88704.9119   339.1  707.01
#Mann= 7 ,-1 , 0
       0     .08       0   59.35     .06       0  188.88     .12       0
  231.46     .06       0  250.26    .045       0   267.3     .06       0
  321.88    .016       0
Bank Sta=250.26,267.3
XS Rating Curve= 0 ,0
Exp/Cntr=0.3,0.1

Type RM Length L Ch R = 1 ,26759   ,112.2,119.1,126.4
XS GIS Cut Line= 3
     2295540.224      393017.959     2295485.537      392678.115
     2295462.099      392654.677
#Sta/Elev= 30
       0  720.81    23.7  718.53    43.5  718.23    47.5  717.89    63.2714.2367
    71.2  712.36    98.9  707.98   106.8  706.09   118.7  702.43   126.6  701.21
   134.5  700.94   193.5 701.058  213.92701.0544   229.5  701.13   233.4  700.74
   237.2  699.79   241.4   699.2   249.3  699.18   253.2  699.48   257.2  700.42
   261.1     701   280.9   701.2   300.7  702.61   324.4  703.23  336.78703.9152
   344.2  704.62   351.6  706.26   362.6  706.71   373.7  706.64   377.4  707.19
#Mann= 7 ,-1 , 0
       0     .08       0    63.2     .06       0   193.5     .12       0
  213.92     .06       0   237.2    .045       0   257.2     .06       0
  336.78    .016       0
#XS Ineff= 2 , 0
          157.12  703.27
Permanent Ineff=
       F       F
Bank Sta=237.2,257.2
XS Rating Curve= 0 ,0
Exp/Cntr=0.3,0.1

Type RM Length L Ch R = 1 ,26639.9 ,88.9,90,89.7
XS GIS Cut Line= 3
     2295588.401       393012.75     2295628.766      392688.531
     2295584.495      392601.292
#Sta/Elev= 30
       0  717.93    35.9  715.16    55.8  714.04    91.8 710.419    99.6  709.98
   107.6  708.99   127.5  705.05   139.4  701.72   143.4  700.84   147.4  700.32
   159.4   699.8   195.2  699.26   235.1  699.43   239.1   699.3     243  698.74
  249.04  697.33     255   696.1     259  696.37  262.52   697.3     267  698.93
   270.9  699.49   290.9  699.23   322.7  700.56   361.9  700.73   377.6  700.42
  387.85700.7431   397.2  701.29     405  702.39   408.9  702.58   424.6   702.4
#Mann= 5 ,-1 , 0
       0     .08       0    91.8     .06       0  249.04    .045       0
  262.52     .06       0  387.85    .016       0
#XS Ineff= 2 , 0
          191.91  701.63
Permanent Ineff=
       F       F
Bank Sta=249.04,262.52
XS Rating Curve= 0 ,0
Exp/Cntr=0.3,0.1

Type RM Length L Ch R = 1 ,26549.9 ,259.1,267.3,274.4
XS GIS Cut Line= 3
     2295673.037      393001.031     2295713.401      392676.813
     2295669.131      392589.573
#Sta/Elev= 30
       0  718.28       8  718.18      12  717.75    39.8  713.31    55.8  712.18
   64.76710.9423    83.7     708   123.5  700.77   131.5  699.73   135.5  699.38
   163.4  698.22   187.3  697.77   223.1  697.73   235.1  698.13     251  698.36
     255  697.66     259   696.3     263  694.92     267  694.78   274.9  695.55
   278.9  696.21   282.9  697.48   286.9  698.14   306.8  698.26   330.6  698.08
   338.5  698.21  372.45699.6031   385.4   700.2   412.8  700.72   424.6  701.33
#Mann= 5 ,-1 , 0
       0     .08       0   64.76     .06       0     259    .045       0
   278.9     .06       0  372.45    .016       0
#XS Ineff= 2 , 0
          189.35  700.33  302.31          699.22
Permanent Ineff=
       F       F
Bank Sta=259,278.9
XS Rating Curve= 0 ,0
Exp/Cntr=0.3,0.1

Type RM Length L Ch R = 1 ,26282.6 ,291,300.7,309.5
XS GIS Cut Line= 2
     2295824.078      393024.469     2295985.537      392672.906
#Sta/Elev= 30
       0  717.65      12  716.42    27.9   714.4    67.8  707.89    83.8  703.35
   115.7  697.32   131.6   694.9   171.5  692.64   191.4  692.68   203.4  692.99
   227.3  692.82  291.58693.6569   311.1  693.69   315.1   693.5  316.82  693.06
     323  691.82     327  691.96     331  692.74  332.22  693.18     335  693.76
   337.7694.7657     339  695.25     343  695.96     351  695.89     355  696.32
   362.9  697.65   366.9  698.03   378.9  698.13   382.9  698.75   386.9  701.66
#Mann= 5 ,-1 , 0
       0     .06       0  291.58     .12       0  316.82    .045       0
  332.22     .12       0   337.7    .016       0
Bank Sta=316.82,332.22
XS Rating Curve= 0 ,0
Exp/Cntr=0.3,0.1

Type RM Length L Ch R = 1 ,25981.9 ,295.3,302.3,306.4
XS GIS Cut Line= 2
     2295986.839      393093.479     2296257.672      392843.479
#Sta/Elev= 30
       0  715.06    31.7  711.74   66.18707.3625    87.2  704.24    91.2  703.28
    99.1  700.28     107  696.28     111  694.71   114.9  694.29   118.9  692.92
   126.8  688.84   138.7  686.99   170.4  688.56   186.3   688.1   198.2  688.33
   206.1  687.13     210  687.03   221.9  688.03   229.9  690.39   241.8  691.38
   245.7  692.01  251.72693.8773   261.6  695.24   277.4  695.41   281.4  696.68
   289.3  701.74  294.23704.1454   309.1  710.94     329  720.71   368.6  741.21
#Mann= 6 ,-1 , 0
       0     .06       0   66.18     .12       0   198.2    .045       0
   221.9     .12       0  251.72    .016       0  294.23     .12       0
Bank Sta=198.2,221.9
XS Rating Curve= 0 ,0
Exp/Cntr=0.3,0.1

Type RM Length L Ch R = 1 ,25679.6 ,329.1,340.4,344.2
XS GIS Cut Line= 3
     2296071.474      393344.781     2296179.547      393273.167
     2296477.724      393079.156
#Sta/Elev= 30
       0  740.21    11.8  738.27    19.6  736.28    35.4  730.66    58.9  720.57
   113.9  694.48   133.6  686.74   153.6   684.5   177.6   683.3   197.6  683.91
   209.6  683.18   249.6  683.15   265.6  682.52   281.5   681.9   289.5  683.08
   293.5  683.72   301.5  683.68   305.5  684.44  310.58687.2014   317.5  691.79
   321.5  693.15   337.5  694.19   341.5  695.62  345.25699.2481   349.5  703.13
   365.5  712.43   401.4  730.65   425.4  741.58   453.4  753.29   485.4  765.42
#Mann= 5 ,-1 , 0
       0     .12       0   265.6    .045       0   289.5     .12       0
  310.58    .016       0  345.25     .12       0
Bank Sta=265.6,289.5
XS Rating Curve= 0 ,0
Exp/Cntr=0.3,0.1

Type RM Length L Ch R = 1 ,25339.2 ,245.8,248.6,249.4
XS GIS Cut Line= 2
     2296133.727      393534.758     2296647.243      393337.097
#Sta/Elev= 30
       0  754.99    27.9  745.21    63.8  730.16    95.7  715.78   139.6   693.9
   147.5  688.96   158.7  680.32   163.5   677.8   167.5  677.19   178.7  678.61
   187.4  679.66   203.4  680.07   227.3  679.79   235.2  678.65   251.2  679.02
   267.2  680.45   279.1  682.41     315  684.15  322.85685.3636   330.9  690.14
   334.9  691.27   350.9  692.09   354.9  694.35  363.59703.2181   394.7  718.67
   434.6  736.11   458.5  744.09   486.4  752.14   530.3  762.07   550.2  767.82
#Mann= 5 ,-1 , 0
       0     .12       0   158.7    .045       0   178.7     .12       0
  322.85    .016       0  363.59     .12       0
Bank Sta=158.7,178.7
XS Rating Curve= 0 ,0
Exp/Cntr=0.3,0.1

Type RM Length L Ch R = 1 ,25090.6 ,298.1,297.6,292.5
XS GIS Cut Line= 2
     2296206.891      393726.292     2296653.506      393593.479
#Sta/Elev= 30
       0  749.96    35.8  734.96    67.7  720.24   127.4  689.61   131.4  687.29
   135.4  684.02   143.4  676.35   147.4  674.48   151.3  674.12   163.3  676.84
   167.3  677.11   183.2  676.74   199.1  677.55     235  675.86   250.9  674.78
   258.9  676.25   278.8  676.72   302.7  680.36   314.6  680.75   318.6  681.64
  322.03683.4493   330.5  687.56   346.5  688.62   350.4  689.51  354.92693.4122
   358.4  696.84   362.4  699.66   386.3  711.13     446  735.99   465.9  742.57
#Mann= 5 ,-1 , 0
       0     .12       0     235    .045       0   258.9     .12       0
  322.03    .016       0  354.92     .12       0
Bank Sta=235,258.9
XS Rating Curve= 0 ,0
Exp/Cntr=0.3,0.1

Type RM Length L Ch R = 1 ,24793   ,277.8,274.8,269.7
XS GIS Cut Line= 2
     2296331.891      393945.042     2296731.631      393790.094
#Sta/Elev= 30
       0  725.63    11.9  724.54    15.9   723.3   23.61718.3511    31.8  712.94
    55.6  698.79    75.4     685    87.3  677.44    91.3  675.49    95.3   674.5
   107.2  673.46   115.1  673.47   157.2  671.17   166.7   669.7   170.7  669.76
   177.2  670.99   182.6  671.83  208.48672.4588   238.2  673.18   247.7 675.636
     266  677.56  279.16678.2908   293.8  678.36   297.7  678.92   301.7  680.87
  306.01683.8166   325.5  692.49   349.3  704.55   381.1  719.24   428.7  739.86
#Mann= 8 ,-1 , 0
       0    .016       0   23.61     .12       0   157.2    .045       0
   177.2     .12       0  208.48     .06       0   247.7     .12       0
  279.16    .016       0  306.01     .12       0
Bank Sta=157.2,177.2
XS Rating Curve= 0 ,0
Exp/Cntr=0.3,0.1

Type RM Length L Ch R = 1 ,24518.2 ,42.8,43,42.8
XS GIS Cut Line= 3
     2296403.723      394179.308     2296500.077      394172.798
     2296828.202      393987.902
#Sta/Elev= 30
       0  730.49    11.6  726.43    30.9  718.83    65.7  706.86    81.1  700.57
    88.8  697.87    96.6  693.88   120.4  678.41   124.3  676.98  129.04676.2831
   148.1  675.16   179.8  671.15  194.48  667.65   195.7  666.94   199.6  666.03
   203.6  665.61   207.6  666.01   215.5  667.82   223.4  668.28     271   668.7
   286.9  670.17   298.8  672.48   306.7  673.55   318.6  673.57   322.6  674.19
   330.5  679.68  347.61687.4886     382  704.26     390  707.47   473.2  743.78
#Mann= 5 ,-1 , 0
       0     .12       0  129.04    .016       0  194.48    .045       0
   215.5    .016       0  347.61     .12       0
Bank Sta=194.48,215.5
XS Rating Curve= 0 ,0
Exp/Cntr=0.3,0.1

Type RM Length L Ch R = 1 ,24475.2 ,136.5,136.2,136.2
XS GIS Cut Line= 3
     2296424.556      394214.465      2296520.91      394207.954
     2296849.035      394023.058
#Sta/Elev= 30
       0  718.26    34.8  707.55    61.8  697.78    92.7  687.28   124.3  678.16
   140.2  674.17   148.1  672.68   175.9  669.88   202.5  665.98   207.6  664.96
   215.5   664.5   219.5  664.64   227.4   666.7   231.4   667.2   255.2  667.48
  265.74 667.966   286.9  670.22   298.8  671.98   306.7   672.5   314.6  672.34
   318.6  673.99   322.6  677.56   326.5  680.38  333.92683.1439   346.3  688.36
   358.2  693.88   366.2  697.08   374.1  701.11   449.4   734.8   473.2  744.35
#Mann= 5 ,-1 , 0
       0     .12       0   202.5    .045       0   227.4     .12       0
  265.74    .016       0  333.92     .12       0
Bank Sta=202.5,227.4
XS Rating Curve= 0 ,0
Exp/Cntr=0.3,0.1

Type RM Length L Ch R = 1 ,24339   ,150.9,151.3,150.8
XS GIS Cut Line= 2
     2296506.587      394369.413     2296923.254      394135.038
#Sta/Elev= 30
       0  708.38    39.8   701.6    71.7  694.29    99.6  686.25   107.6  683.54
   115.5  679.18   119.5  677.44   135.4  671.46   143.4  671.01   155.4  667.92
   187.2  666.78   215.1  667.39   219.1  666.91   222.8  665.55   227.1  663.89
   231.1  663.51     239  663.59     247   664.6     259  664.87  283.06666.5558
   294.8  667.68   306.8  667.83  311.84 670.345   314.7  672.44   318.7  674.56
   346.6  687.31   374.5   701.3   390.4  709.93   414.3   721.6   478.1  747.76
#Mann= 5 ,-1 , 0
       0     .12       0   222.8    .045       0     247     .12       0
  283.06    .016       0  311.84     .12       0
Bank Sta=222.8,247
XS Rating Curve= 0 ,0
Exp/Cntr=0.3,0.1

Type RM Length L Ch R = 1 ,24187.7 ,64.9,64.8,65.2
XS GIS Cut Line= 2
     2296588.618      394491.808     2297005.285      394257.433
#Sta/Elev= 30
       0  724.04    35.8  711.14   119.5  675.84   135.4  669.88   143.4  667.31
   155.4   664.5   167.3  662.68   195.2  662.67   203.2  663.14   208.4  662.66
   219.1  660.95   231.1  662.57     243  663.57     255  663.87  260.96665.0029
   266.9  666.48   282.8  667.31   290.8  666.94   294.8  667.22  300.56669.9368
   306.8  672.35   314.7  676.08   338.6  688.45   354.6  697.92   374.5  708.79
   418.3  729.97   442.2  740.44   458.1  746.26   470.1  749.97   478.1  752.99
#Mann= 5 ,-1 , 0
       0     .12       0   208.4    .045       0   231.1     .12       0
  260.96    .016       0  300.56     .12       0
#XS Ineff= 2 , 0
          167.52  672.12  282.41          670.46
Permanent Ineff=
       F       F
Bank Sta=208.4,231.1
XS Rating Curve= 0 ,0
Exp/Cntr=0.3,0.1

Type RM Length L Ch R = 1 ,24122.9 ,31,30.9,31
XS GIS Cut Line= 2
     2296628.202      394540.767     2297044.868      394306.392
#Sta/Elev= 30
       0  720.58    27.9  709.93    79.7  686.99    83.7  684.92    87.6  681.96
    95.6  673.73    99.6  671.84   103.4 671.517   127.5  671.39  141.02 668.939
   151.4  666.66  177.27665.0315  200.46665.8987   211.1  666.01   215.1  664.59
   223.1  660.97   227.1   660.9     235   664.8  238.22665.9672   278.9  667.21
  290.16669.2224   298.8  671.12   302.8  672.74   314.7  682.68   326.7  689.51
   362.5  708.43   370.5  711.85   422.3  737.77   458.1  753.09   478.1  759.71
#Mann= 9 ,-1 , 0
       0     .12       0   103.4     .08       0  141.02     .12       0
  177.27     .08       0  200.46     .12       0   215.1    .045       0
     235     .12       0  238.22    .016       0  290.16     .12       0
#XS Ineff= 2 , 0
          200.26  668.93
Permanent Ineff=
       F       F
Bank Sta=215.1,235
XS Rating Curve= 0 ,0
Exp/Cntr=0.3,0.1

Type RM Length L Ch R = 1 ,24092   ,211.7,212.2,211.3
XS GIS Cut Line= 2
     2296648.514      394563.683     2297065.181      394329.308
#Sta/Elev= 30
       0  717.65    47.8  697.64    75.7  684.94    79.7  682.69    87.6  674.08
    91.6  671.68    95.9 670.983   115.5  670.91  150.96665.9751   175.3   664.6
   207.2   664.7   211.1  664.06   219.1  660.25   223.1   660.5  229.78  663.98
     235  666.22  251.63666.2826   274.9  666.24   278.9  667.81  283.73671.2738
   290.8  675.43   306.8  678.94   310.7  681.05   318.7   688.2   326.7  693.73
   338.6   698.7   358.6  710.44   422.3   740.8   458.1  756.19   478.1  762.84
#Mann= 7 ,-1 , 0
       0     .12       0    95.9     .08       0  150.96     .12       0
   211.1    .045       0  229.78     .08       0  251.63    .016       0
  283.73     .12       0
Bank Sta=211.1,229.78
XS Rating Curve= 0 ,0
Exp/Cntr=0.3,0.1

Type RM Length L Ch R = 1 ,23879.8 ,294.5,292.5,289.6
XS GIS Cut Line= 4
     2296671.917       394720.34      2296793.12      394723.567
     2296956.417      394631.712     2297132.114      394531.379
#Sta/Elev= 30
       0     730      43  715.67   121.2  690.88   157.1   677.2   165.1  673.29
   173.1  666.93     177  664.35  182.15663.3738     189  662.73     197  659.38
     201  658.82   276.7  658.28  292.12658.6967   296.6  659.27   298.6  659.03
   308.6  657.11   318.6  658.57   328.4  662.05   332.4  662.92   344.3  663.56
   348.3  664.24   352.2  667.16  357.64673.0632   360.2   675.7   364.2  678.56
     376  684.94   419.7  706.24   467.3  730.85   491.1  742.28   510.9     750
#Mann= 6 ,-1 , 0
       0     .12       0  182.15     .06       0  292.12     .12       0
   298.6    .045       0   318.6    .016       0  357.64     .12       0
Bank Sta=298.6,318.6
XS Rating Curve= 0 ,0
Exp/Cntr=0.3,0.1

Type RM Length L Ch R = 1 ,23587.3 ,169.4,169.7,169.4
XS GIS Cut Line= 3
     2296868.876      395042.048     2297156.114      394838.691
     2297239.772      394764.537
#Sta/Elev= 30
       0  724.01      16  719.49      32  713.86      60  701.66      76  691.88
      88   689.5      92  687.89     112  674.49     124     665     128   663.1
  143.69658.9382     156  658.72     176  655.95  189.98655.5807     244  653.49
  270.19654.1764   283.5   654.3     288  654.17     296  652.41     300  652.49
   303.5   654.2   307.9  657.87   311.9  658.94   323.9  659.18   327.9  660.46
  337.35671.0885   339.9  673.46   351.9     680   435.8  716.76   463.7     730
#Mann= 7 ,-1 , 0
       0     .12       0  143.69    .016       0  189.98     .06       0
  270.19     .12       0   283.5    .045       0   303.5    .016       0
  337.35     .12       0
Bank Sta=283.5,303.5
XS Rating Curve= 0 ,0
Exp/Cntr=0.3,0.1

Type RM Length L Ch R = 1 ,23417.6 ,322,293.6,261.8
XS GIS Cut Line= 4
     2296920.422      395091.572     2297053.631      395102.363
     2297281.439      394947.357      2297307.25       394848.33
#Sta/Elev= 30
       0  711.58     3.9  710.36    15.7  704.14    51.1  690.01    74.7  677.88
   82.24672.7516    90.4  664.66    94.3  661.94    98.3  660.54  130.55658.4285
   149.6  655.36   157.6  654.66   225.5  654.56   241.5  651.86   268.9  651.24
   281.4  649.56   285.4  650.21   288.9  651.49   293.4  652.65   305.4  652.86
   317.3  654.07   369.2  655.62  383.65657.7314  388.19658.1693   413.1  658.18
   417.1  659.99  424.99666.0987   440.7  673.96   487.9  701.75   511.5  714.44
#Mann= 8 ,-1 , 0
       0     .12       0   82.24     .06       0  130.55     .12       0
   268.9    .045       0   288.9     .06       0  383.65     .12       0
  388.19    .016       0  424.99     .12       0
Bank Sta=268.9,288.9
XS Rating Curve= 0 ,0
Exp/Cntr=0.3,0.1

Type RM Length L Ch R = 1 ,23124.1 ,118,114,108.3
XS GIS Cut Line= 4
     2297324.501       395266.87     2297387.375      395134.456
     2297347.439      394949.681     2297347.375      394883.792
#Sta/Elev= 30
       0  701.43    15.8  698.42    27.7  695.67    55.5  686.63    91.1  671.73
   138.7  653.22   146.6  651.77   158.4  648.46   162.3  647.89   174.2  647.52
   177.6  646.97     186   645.2   193.8  645.06   201.7  646.56   205.7  647.03
   217.5  647.03   229.3  647.77   237.2  647.48     245  647.98   256.9  647.98
  270.99648.8049  297.27652.4183   304.1  653.07     312   656.1   315.9  656.84
   335.6  657.03  338.44 658.734   347.2  665.75   358.9  671.88   401.5  696.45
#Mann= 6 ,-1 , 0
       0     .12       0   177.6    .045       0   201.7     .12       0
  270.99     .06       0  297.27    .016       0  338.44     .12       0
Bank Sta=177.6,201.7
XS Rating Curve= 0 ,0
Exp/Cntr=0.3,0.1

Type RM Length L Ch R = 1 ,23010.1 ,209.3,231.8,253.8
XS GIS Cut Line= 3
     2297590.397      395294.789     2297428.087      394940.928
     2297425.831      394877.426
#Sta/Elev= 30
       0  677.65    23.8  670.52    39.7  666.72    87.4  657.56   107.3  655.95
   115.2   654.4   135.1  652.13   158.9  651.15   178.8  649.56   222.5  649.73
   246.3  647.01   274.1  646.69     282  645.23     294   643.2   297.9  643.53
   305.9  645.52   309.9  645.91  320.24645.5173  328.61645.7281   353.6  649.42
  363.96654.1049   369.4  655.19   385.3  654.96   389.3   657.8  394.25662.5942
   397.2  665.34   401.2  668.13   417.1  677.46   440.9  692.62   452.8  699.59
#Mann= 7 ,-1 , 0
       0     .12       0     282    .045       0   305.9     .12       0
  320.24     .06       0  328.61     .12       0  363.96    .016       0
  394.25     .12       0
Bank Sta=282,305.9
XS Rating Curve= 0 ,0
Exp/Cntr=0.3,0.1

Type RM Length L Ch R = 1 ,22778.2 ,71.1,70.7,71
XS GIS Cut Line= 4
     2297629.179      395237.602     2297574.344      395138.307
     2297705.292      394887.359     2297696.114      394825.664
#Sta/Elev= 30
       0     670    27.4     664    50.8  659.61    74.3  655.73      86  652.02
      90  651.16  117.62649.7652     151647.1937  203.91645.0593  222.38644.3884
  255.46643.7601   288.8     643   308.8  644.02   312.8  643.87   320.7  641.85
   324.7  641.91   328.7  643.24  330.55  644.29   340.7   649.1   344.7  649.95
   360.6  650.96   372.6  650.94   376.6  651.81   392.5  657.78  394.39658.8337
   396.5  660.01   400.4  663.46   408.2  671.98   412.1  675.79   458.9     700
#Mann= 9 ,-1 , 0
       0     .12       0  117.62     .06       0     151     .12       0
  203.91    .016       0  222.38     .06       0  255.46     .12       0
   312.8    .045       0  330.55    .016       0  394.39     .12       0
Bank Sta=312.8,330.55
XS Rating Curve= 0 ,0
Exp/Cntr=0.3,0.1

Type RM Length L Ch R = 1 ,22707.5 ,119.8,105.4,89
XS GIS Cut Line= 4
     2297701.005      395251.829     2297646.171      395152.534
     2297777.118      394901.587     2297767.941      394839.891
#Sta/Elev= 30
       0  682.67    39.1  671.22   60.57665.9565    78.2  661.48   87.47660.2126
   105.6  657.71     123 651.302   129.4  649.76  140.98649.3433   149.3  648.75
   165.3  645.82  177.89645.4793     229  643.53   284.9  643.21   290.3  641.38
   296.8  639.26   310.3  641.13  318.07641.5565   336.7  641.43   352.6   645.1
   360.6  644.87  368.46647.9798   384.5  651.67   412.1  652.68  420.83656.9001
   431.6  660.72   435.5  663.42   443.3  670.46     455  682.84   458.9   685.1
#Mann= 11 ,-1 , 0
       0     .12       0   60.57     .06       0   87.47     .12       0
     123     .06       0  140.98    .016       0  177.89     .06       0
   290.3    .045       0   310.3     .06       0  318.07     .12       0
  368.46    .016       0  420.83     .12       0
Bank Sta=290.3,310.3
XS Rating Curve= 0 ,0
Exp/Cntr=0.3,0.1

Type RM Length L Ch R = 1 ,22602.2 ,145.5,151.8,158
XS GIS Cut Line= 3
     2297847.346       395171.77     2297843.299      395081.354
     2297812.114       394822.01
#Sta/Elev= 30
       0  679.97    35.4     667    47.2  663.32    55.1  661.95      59  660.57
    66.9  656.28    70.8  654.79    78.7  654.05   84.36652.5064    98.4  646.81
   110.3  642.95   126.1  639.99     138  639.26   157.8  639.64   197.4  639.08
   207.3  638.31   217.2  637.31   221.1  637.41   227.3  638.59   256.7  642.29
   260.7  643.46  271.04649.8881   276.5  651.61   284.4  652.48   296.3  652.84
  303.37655.7512   308.2  658.41   320.1  670.59     324  673.71   351.7     690
#Mann= 6 ,-1 , 0
       0     .12       0   84.36     .06       0   207.3    .045       0
   227.3     .12       0  271.04    .016       0  303.37     .12       0
Bank Sta=207.3,227.3
XS Rating Curve= 0 ,0
Exp/Cntr=0.3,0.1

Type RM Length L Ch R = 1 ,22450.3 ,257.7,243.3,228.8
XS GIS Cut Line= 4
     2297912.114      395187.973     2297964.168       395084.59
     2297990.678      394879.102      2297945.66      394794.082
#Sta/Elev= 30
       0     680    47.9   667.7    63.9  665.47    67.8  664.44    79.8  660.33
    87.8  655.98    91.8  654.63   103.8   653.2   119.7     649   139.6  644.77
   179.5  639.01   211.4  636.42   223.3  636.63   231.3  634.67   235.3   634.3
   243.3  636.36   263.2  637.24   283.1  637.38  299.02638.3919   330.6  640.63
     346   644.6  349.55646.3477   357.6  652.15   365.3  653.24   380.7  653.25
   384.5  654.37  386.91655.7542   392.2  659.88   399.9  667.93   419.1     680
#Mann= 6 ,-1 , 0
       0     .12       0   223.3    .045       0   243.3     .06       0
  299.02     .12       0  349.55    .016       0  386.91     .12       0
Bank Sta=223.3,243.3
XS Rating Curve= 0 ,0
Exp/Cntr=0.3,0.1

Type RM Length L Ch R = 1 ,22207   ,191.1,194.9,198.4
XS GIS Cut Line= 3
     2298260.898      395060.496     2298240.378      394992.114
     2298119.861      394741.816
#Sta/Elev= 30
       0     681    15.9  675.22    47.6  662.22   103.1  635.87   110.1  634.46
   111.1  634.31     115  632.67     119  631.78     123  631.91   130.1  633.77
   134.9  634.23  140.46 634.066   158.7  633.45   190.4  633.22   198.4  633.49
   210.3  633.14   222.2  633.76  241.87 635.477   257.9  636.88   281.7  640.57
   293.6  643.87   297.6  645.96  299.49647.2925   305.5  651.65   309.5  652.66
   325.4  653.34   329.4  655.46   333.3  659.65  336.31661.5538   349.2  668.38
#Mann= 7 ,-1 , 0
       0     .12       0   110.1    .045       0   130.1     .12       0
  140.46     .06       0  241.87     .12       0  299.49    .016       0
  336.31     .12       0
Bank Sta=110.1,130.1
XS Rating Curve= 0 ,0
Exp/Cntr=0.3,0.1

Type RM Length L Ch R = 1 ,22012.1 ,192.1,192.3,191.6
XS GIS Cut Line= 3
     2298420.696      394956.537     2298331.644      394672.066
      2298279.43      394631.854
#Sta/Elev= 30
       0     670    51.7  652.14    63.6  646.25    75.5  641.16   100.2   629.7
   107.3   628.9   120.2     630   143.1  630.86  151.88630.3616  159.39630.1276
   178.8  630.27   186.8  629.23   190.8  629.13   194.8  630.54   202.7  635.19
   206.7  637.02   210.6  638.24   222.6  640.19  233.16642.5679   242.4  646.63
   258.3  647.44   262.3  649.48   265.6652.3923   270.3  656.41   274.2  658.58
   282.2  661.89   298.1     670   313.6   674.4   344.6  684.97     364     690
#Mann= 7 ,-1 , 0
       0     .12       0   100.2    .045       0   120.2     .12       0
  151.88     .06       0  159.39     .12       0  233.16    .016       0
   265.6     .12       0
Bank Sta=100.2,120.2
XS Rating Curve= 0 ,0
Exp/Cntr=0.3,0.1

Type RM Length L Ch R = 1 ,21819.8 ,61.8,63.6,65.3
XS GIS Cut Line= 4
     2298533.928      394906.725      2298571.04      394822.538
     2298521.804      394669.696     2298455.794      394629.819
#Sta/Elev= 30
       0     660    15.3  656.06    26.8  651.42    38.3  645.73    53.7  641.53
    65.2  636.32      69  635.41    72.8  634.81    88.2  633.99    99.8  631.69
   115.5  629.73   127.2  629.02   146.8  629.22   157.5  627.62   166.4  626.03
   170.3  626.01   177.5  627.28   197.8   628.8   209.5  629.07     216630.1266
   225.2  632.25   240.8  632.76   244.8  634.32   248.7   636.6  251.69637.3666
   264.2  640.53   275.7  644.59     295  650.33   310.4  655.67   329.7  661.21
#Mann= 5 ,-1 , 0
       0     .12       0   157.5    .045       0   177.5     .12       0
     216    .016       0  251.69     .12       0
Bank Sta=157.5,177.5
XS Rating Curve= 0 ,0
Exp/Cntr=0.3,0.1

Type RM Length L Ch R = 1 ,21756.2 ,264.1,298.7,331.9
XS GIS Cut Line= 4
     2298591.616      394915.155       2298636.7       394839.64
     2298583.534      394646.963     2298478.581      394588.586
#Sta/Elev= 30
       0  644.29       8  641.43      16  639.27   19.75  637.77      28  633.59
      32   632.5      44  632.31      56  630.43      76  629.78   131.9  626.66
  156.58626.6617   187.9   626.9   197.7  626.42   207.9  625.24   217.7  626.33
   227.9  626.43  235.36626.9681   255.8  628.91   267.8  629.05  275.45629.6385
  309.15  630.83   345.9  631.35   349.8  633.17   353.7  635.98   357.6  638.11
  361.88639.8381   369.2  642.99   384.7  648.12   400.2   654.1   407.9  656.29
#Mann= 9 ,-1 , 0
       0     .12       0   19.75     .06       0  156.58     .12       0
   197.7    .045       0   217.7     .12       0  235.36    .016       0
  275.45     .12       0  309.15     .08       0  361.88     .12       0
Bank Sta=197.7,217.7
XS Rating Curve= 0 ,0
Exp/Cntr=0.3,0.1

Type RM Length L Ch R = 1 ,21457.5 ,180.4,183.4,186.8
XS GIS Cut Line= 2
     2298605.534      394944.489      2298934.31      394770.878
#Sta/Elev= 30
       0   641.9       8  637.72      20  632.84   22.89632.4426      32  631.82
      40  630.72      72  628.82   127.9   627.6   191.9  622.94   211.6  622.51
   223.9  621.18  230.04  623.06  238.99628.4995   243.9  629.97   247.9  630.45
   259.9  630.85  278.69630.7451   287.8  631.26   299.8  631.22   303.8  631.82
   307.8  633.66   315.8  640.32   327.8  648.48   331.8  651.71   335.8  654.45
   339.8  655.71  344.63655.6111   359.8  655.08   363.8  655.93   371.8  658.58
#Mann= 7 ,-1 , 0
       0     .12       0   22.89     .06       0   211.6    .045       0
  230.04     .06       0  238.99    .016       0  278.69     .12       0
  344.63    .016       0
Bank Sta=211.6,230.04
XS Rating Curve= 0 ,0
Exp/Cntr=0.3,0.1

Type RM Length L Ch R = 1 ,21274.1 ,388.9,393.3,394.9
XS GIS Cut Line= 3
      2298589.91      395114.332      2298938.47      394984.537
     2299021.164      394984.537
#Sta/Elev= 30
       0     670      16     662      44  646.52      52     641      56  638.89
      64  636.39      72   632.6      76  631.62      92   631.3     112  626.73
  147.05624.1789     200  621.92     244  621.32     260  620.21   290.2  620.63
     300  618.69     304  618.63   310.2  621.68     316  624.72  324.92 626.219
   351.9  628.24   355.9  629.24  360.88634.5978   367.9  645.25   371.9     650
   379.8  653.82   391.6  657.75   403.4  660.74   442.8  668.69   454.6     670
#Mann= 6 ,-1 , 0
       0     .12       0  147.05     .06       0   290.2    .045       0
   310.2     .06       0  324.92    .016       0  360.88     .12       0
Bank Sta=290.2,310.2
XS Rating Curve= 0 ,0
Exp/Cntr=0.3,0.1

Type RM Length L Ch R = 1 ,20880.8 ,277.9,279.2,280.2
XS GIS Cut Line= 2
     2298687.468      395419.044      2299130.68      395284.537
#Sta/Elev= 30
       0  675.13    47.9   654.1    79.9   637.9    95.8  629.04   107.8  626.61
   127.8   620.5  149.99617.4294   171.7  616.41   183.7  615.03   195.6   616.2
   223.6  616.63   243.6  615.71   251.6  616.28   263.5  615.83   268.6 616.411
  273.74 618.234   283.5  620.59  304.44621.5611   315.4  621.23  335.13622.5989
   343.4  625.99   347.4   626.5   359.2626.3115   367.3     628   371.3  630.43
   383.3  640.51   387.3  643.33   399.3  649.99   439.2  669.72   463.2     680
#Mann= 9 ,-1 , 0
       0     .12       0  149.99     .06       0   171.7    .045       0
   195.6     .12       0   268.6     .06       0  273.74     .08       0
  304.44     .12       0  335.13    .016       0   359.2     .12       0
Bank Sta=171.7,195.6
XS Rating Curve= 0 ,0
Exp/Cntr=0.3,0.1

Type RM Length L Ch R = 1 ,20601.6 ,307.1,304.9,301.4
XS GIS Cut Line= 2
     2298707.144      395680.383     2299175.379      395572.537
#Sta/Elev= 30
       0  705.03    67.5  680.36   103.2  665.79     139  649.16   154.9  639.61
   166.8   630.4   174.7  622.88   186.6  614.14   190.6  612.28   194.6   611.5
   218.4   613.9   234.3   614.2   254.2  612.94   262.1  611.45   266.1   611.2
   277.1  613.76   285.9  614.97  299.51615.6169   317.7  616.64   329.6  616.86
   337.5  616.35  344.01617.2759   349.4  618.31  374.19621.3083   385.2   622.7
   397.1  623.39   436.8  624.21   444.8  625.61   452.7  628.37   480.5     630
#Mann= 6 ,-1 , 0
       0     .12       0   254.2    .045       0   277.1     .12       0
  299.51     .08       0  344.01    .016       0  374.19     .12       0
Bank Sta=254.2,277.1
XS Rating Curve= 0 ,0
Exp/Cntr=0.3,0.1

Type RM Length L Ch R = 1 ,20296.7 ,323.8,327.6,328.8
XS GIS Cut Line= 3
     2298796.243      395944.666     2298911.844      395952.537
     2299294.623      395816.537
#Sta/Elev= 30
       0     680      40  660.53    59.9  649.95    83.9  636.34    95.9  630.19
   107.9  624.89   115.9     620   127.8   615.8   143.8  611.67   159.7  609.91
   175.6  609.63   191.5  610.41   219.4  609.12   236.4   609.3   247.3  607.77
   251.3  607.78   259.2  609.63  269.14612.2382  290.88613.0117     307  611.21
  322.02612.2808   342.9   613.2  354.48614.4556   386.7  619.37   426.5  624.63
  447.01626.1573   466.3  628.36  473.33631.0332   498.2  639.43   522.1     650
#Mann= 9 ,-1 , 0
       0     .12       0   236.4    .045       0   259.2     .12       0
  269.14    .016       0  290.88     .08       0  322.02     .06       0
  354.48    .016       0  447.01     .06       0  473.33     .12       0
#XS Ineff= 2 , 0
                          286.52          616.12
Permanent Ineff=
       F       F
Bank Sta=236.4,259.2
XS Rating Curve= 0 ,0
Exp/Cntr=0.3,0.1

Type RM Length L Ch R = 1 ,19969.1 ,317.3,315.1,310.4
XS GIS Cut Line= 3
     2298850.952      396279.375     2298929.234      396235.416
     2299333.044      396132.537
#Sta/Elev= 30
       0  659.99    31.2  647.79    66.4  631.66    85.9  621.58    97.7  617.23
   113.6  612.51   125.5  609.98   153.3  607.57   165.2  604.36   173.1  603.78
     189  604.29   204.9  606.27   216.8  606.79   232.6  605.27   252.5  606.62
   256.5  607.95   264.4  613.14   270.7 614.848   288.2  615.74  307.89615.2526
     312  616.05     316  618.77   327.9  632.75   331.9  634.98  338.23636.5974
   371.6  640.86   423.2  645.73   450.9  650.75   486.6  655.85   506.5     660
#Mann= 6 ,-1 , 0
       0     .12       0   165.2    .045       0     189     .12       0
   270.7    .016       0  307.89     .08       0  338.23     .12       0
Bank Sta=165.2,189
XS Rating Curve= 0 ,0
Exp/Cntr=0.3,0.1

Type RM Length L Ch R = 1 ,19654   ,280.8,280.8,279.1
XS GIS Cut Line= 3
     2298929.799      396502.223     2299002.551        396530.1
     2299381.585      396386.008
#Sta/Elev= 30
       0     650    66.2  633.28    81.9  628.72   105.7  618.73   125.6   608.5
   141.5  603.54   165.4  602.98   181.3  601.83   193.2  602.44   205.1  601.31
     221  602.81     229  602.09     233  600.82   240.9  600.16   252.8  602.31
  262.23603.3272   272.7  605.45   288.6  614.26   292.6  615.16  303.01615.1686
   332.3   615.3   336.3  616.35  338.74618.7656   344.3  625.88   348.2  630.01
   352.2  632.34     380  639.04   407.9  646.88   459.6  661.79   483.4     670
#Mann= 6 ,-1 , 0
       0     .12       0     229    .045       0   252.8     .12       0
  262.23     .06       0  303.01    .016       0  338.74     .12       0
Bank Sta=229,252.8
XS Rating Curve= 0 ,0
Exp/Cntr=0.3,0.1

Type RM Length L Ch R = 1 ,19373.2 ,306.3,308.6,309.8
XS GIS Cut Line= 3
     2299021.743      396766.012     2299154.112      396763.328
     2299515.365      396616.152
#Sta/Elev= 30
       0  637.13      35  631.44    62.3  625.24     109   611.3   116.8  609.61
   148.3  606.65   160.3  604.24   172.2   604.8   188.1  603.56     204  598.97
     224  599.12   247.8  597.74  258.62598.2874     263  597.78   267.7   596.6
   275.7  596.38   279.7  597.38     283  599.65  286.63602.5825   295.6  609.43
   299.6  611.13   315.5  612.64  334.83611.9357   359.3  611.97   363.3  612.91
   367.2  615.17   383.2  628.25   403.1  639.88   482.7  681.65   522.5  700.64
#Mann= 6 ,-1 , 0
       0     .12       0  258.62     .06       0     263    .045       0
     283     .06       0  286.63    .016       0  334.83     .12       0
Bank Sta=263,283
XS Rating Curve= 0 ,0
Exp/Cntr=0.3,0.1

Type RM Length L Ch R = 1 ,19064.6 ,346,346.4,343.6
XS GIS Cut Line= 3
     2299154.241      397038.664     2299237.407       397041.83
     2299617.379      396915.273
#Sta/Elev= 30
       0     630    43.6  624.41    63.4  618.21    91.2  606.98     111  601.98
   126.8  600.55   142.7  597.24   150.6  596.34   174.4  596.33   178.4  595.61
   190.3  594.01   202.7  595.34     218  595.91   233.9   594.5   241.8  596.07
  244.35597.3578  246.48598.5915   253.7   603.9   261.7  607.92  271.94609.2019
   305.3  610.11   309.2  611.56   313.2  615.07  318.09 620.694   325.1  630.62
   329.1  635.24     333  637.98   344.9  643.48   428.2  672.91   483.7     690
#Mann= 7 ,-1 , 0
       0     .12       0   178.4    .045       0   202.7     .06       0
  244.35     .12       0  246.48     .06       0  271.94    .016       0
  318.09     .12       0
Bank Sta=178.4,202.7
XS Rating Curve= 0 ,0
Exp/Cntr=0.3,0.1

Type RM Length L Ch R = 1 ,18718.2 ,247,247.2,242
XS GIS Cut Line= 3
     2299202.175      397370.598     2299590.853      397219.276
     2299727.801       397240.85
#Sta/Elev= 30
       0     630    87.4  625.85    99.3  624.67   111.2  622.37   119.2  619.96
   131.1  615.36     151   605.5   158.9  600.26   166.8  593.88   170.8  591.99
   174.8  591.53   186.7  592.87   202.6  593.56   222.4   592.6   242.3  593.31
   262.2  591.94     294  592.33   305.9  590.47   313.8  591.05  316.54  592.46
  321.04595.9115   325.7  598.68  333.21600.0391   349.6  601.45   369.4  601.69
   401.2  604.46  435.23616.8881   452.8  623.23   492.4  638.82   555.7     660
#Mann= 6 ,-1 , 0
       0     .12       0     294    .045       0  316.54     .06       0
  321.04     .12       0  333.21    .016       0  435.23     .12       0
Bank Sta=294,316.54
XS Rating Curve= 0 ,0
Exp/Cntr=0.3,0.1

Type RM Length L Ch R = 1 ,18471   ,265.4,266.2,266.6
XS GIS Cut Line= 2
     2299307.605      397581.046     2299757.519      397383.132
#Sta/Elev= 30
       0     640      56  627.68    95.9  615.86   147.9  594.78   159.8  589.02
   163.8     588   167.8  587.67   175.8  589.14   191.8  589.82   231.8   589.8
  244.73590.4865   251.8  590.67   255.8  589.89   263.7  587.14   267.7  586.68
   275.7  587.36   285.5   589.5   299.7  593.18  304.91593.8729   319.7  594.85
   335.7  594.52   339.7  595.62   367.6  611.48   388.5612.0875   395.6  613.99
   399.6  616.13   411.6  625.53  420.52629.9474   451.6  642.23   491.5  660.01
#Mann= 7 ,-1 , 0
       0     .12       0  244.73     .06       0   255.8    .045       0
   285.5     .06       0  304.91    .016       0   388.5     .06       0
  420.52     .12       0
Bank Sta=255.8,285.5
XS Rating Curve= 0 ,0
Exp/Cntr=0.3,0.1

Type RM Length L Ch R = 1 ,18204.8 ,252.6,253.7,254.8
XS GIS Cut Line= 3
     2299414.277      397831.075     2299442.503      397804.232
     2299892.837      397618.829
#Sta/Elev= 30
       0  668.57    19.5  663.72    46.9  654.36    86.8  635.88   114.8  619.45
   150.7  592.45   158.7  588.59   198.6  585.48   210.6  586.88  234.55586.6105
   246.5  586.74   258.5  584.22   266.5  585.05   270.5   586.5   278.5  590.01
  282.06 590.439   306.4  591.19  321.97589.8494   330.4   587.9   338.3  587.66
   366.3  589.72   378.3  592.44  391.09600.8052   398.2  604.62  431.15607.3998
   434.2  608.78   446.1  618.08   450.1  620.22     498  641.16     526  652.31
#Mann= 8 ,-1 , 0
       0     .12       0  234.55     .06       0   246.5    .045       0
   270.5     .06       0  282.06    .016       0  321.97     .12       0
  391.09    .016       0  431.15     .12       0
#XS Ineff= 2 , 0
                          296.53          597.09
Permanent Ineff=
       F       F
Bank Sta=246.5,270.5
XS Rating Curve= 0 ,0
Exp/Cntr=0.3,0.1

Type RM Length L Ch R = 1 ,17951.1 ,319.4,350.4,347.7
XS GIS Cut Line= 3
     2299459.656       397983.12     2299584.506      398012.284
     2299952.074       397879.83
#Sta/Elev= 30
       0  665.86   10.23661.6219    62.2  637.56   128.2  602.03   168.1   584.9
     204   582.9   215.9  584.34  251.59584.4863   267.8  585.08   272.2  584.44
   275.7  582.83   283.7  582.04   292.2  583.68   299.6  587.36   303.6   588.3
  315.32588.8058  342.57587.8745   355.5  586.86   363.4  587.43   383.4  597.48
   407.3  599.12   411.3  600.39   419.2  606.64   423.2  608.96   443.2  615.38
  467.34620.3834   475.1  621.82     495  623.05  513.36629.9526   518.9  631.77
#Mann= 9 ,-1 , 0
       0    .016       0   10.23     .12       0  251.59     .06       0
   272.2    .045       0   292.2     .12       0  315.32    .016       0
  342.57     .12       0  467.34    .016       0  513.36     .12       0
#XS Ineff= 2 , 0
                          314.25          592.12
Permanent Ineff=
       F       F
Bank Sta=272.2,292.2
XS Rating Curve= 0 ,0
Exp/Cntr=0.3,0.1

Type RM Length L Ch R = 1 ,17600.7 ,331.7,321.3,308.2
XS GIS Cut Line= 3
     2299520.395      398232.817     2299890.607      398150.044
     2299997.093      398179.559
#Sta/Elev= 30
       0     640    43.9  616.21    67.9  605.84    83.9  600.64   111.8  593.13
   123.8  588.52   139.8  583.43   147.8  579.83   163.7  581.55   172.1  581.02
   183.7  579.07   191.7  579.54   195.7  580.97   199.7  582.31   203.6  582.77
   223.6  581.86   235.6  583.35   280.8586.4297   299.5  587.08  310.27588.8685
  316.04588.9662   327.4  587.56   355.4  585.91   359.4  586.26  367.74 590.155
   387.2  606.37   395.1   611.5   399.1  612.96   458.3   625.5   489.8  629.99
#Mann= 7 ,-1 , 0
       0     .12       0   172.1    .045       0   195.7     .12       0
   280.8     .06       0  310.27     .12       0  316.04    .016       0
  367.74     .12       0
Bank Sta=172.1,195.7
XS Rating Curve= 0 ,0
Exp/Cntr=0.3,0.1

Type RM Length L Ch R = 1 ,17279.3 ,367.8,365.2,360.3
XS GIS Cut Line= 2
     2299742.448      398542.203     2300108.114      398253.096
#Sta/Elev= 30
       0     630    27.9  618.22    39.8  612.46    51.8   607.9    83.7  596.56
    99.6  591.51   107.6  589.61   111.6  588.02   123.5  579.63   129.5  578.06
   143.4  577.12   149.5  578.03   155.4  578.76   171.3  579.28   211.2  578.09
  269.71  579.42   278.9  579.85  295.36582.2512  328.09581.7247   330.7  581.94
   334.7  584.23   342.6  593.84   350.6  602.39   354.6  605.59   366.5  612.39
   386.5  621.01   402.4  626.84   430.3  638.12   454.2  646.55   466.2     650
#Mann= 6 ,-1 , 0
       0     .12       0   129.5    .045       0   149.5     .12       0
  269.71     .06       0  295.36    .016       0  328.09     .12       0
Bank Sta=129.5,149.5
XS Rating Curve= 0 ,0
Exp/Cntr=0.3,0.1

Type RM Length L Ch R = 1 ,16914.1 ,95.1,94.6,94.6
XS GIS Cut Line= 2
     2299990.311      398800.402     2300332.114      398429.856
#Sta/Elev= 30
       0  617.39    43.7  607.26   150.8  594.36   178.6  587.42   186.6  584.43
   202.4  576.72   210.4  575.14   220.7  575.26   234.2   574.1   240.7   575.6
  240.96575.7189   246.1  577.69   250.1  578.06     262  577.12   269.9  575.32
  291.73  577.07   309.6  577.92  332.82 576.578   365.2  573.95   369.2  574.29
  376.86577.6794     385  581.06     393  582.37   404.9   581.9   412.8  582.57
  417.56584.7097   424.7  590.22   436.6  602.24   444.6  607.49   504.1  634.69
#Mann= 8 ,-1 , 0
       0     .12       0   220.7    .045       0   240.7     .12       0
  240.96     .06       0  291.73    .016       0  332.82     .12       0
  376.86    .016       0  417.56     .12       0
#XS Ineff= 2 , 0
                          255.71          581.25
Permanent Ineff=
       F       F
Bank Sta=220.7,240.7
XS Rating Curve= 0 ,0
Exp/Cntr=0.3,0.1

Type RM Length L Ch R = 1 ,16819.5 ,248.9,250.3,241.1
XS GIS Cut Line= 2
     2300067.134      398858.996     2300407.251      398483.358
#Sta/Elev= 30
       0  641.68      16  637.64    31.9  631.76    51.9  629.36    91.8  619.96
   131.7  608.71   143.6  604.25   147.6  601.82   155.6  594.23   171.6  592.74
   175.6  591.26   191.5  578.11   195.5  575.64   199.5   574.5   215.5   573.3
   231.4  572.11   243.4  573.66   255.4  576.42  280.15576.6843  313.23576.0028
   351.1  572.89   375.1  575.44   379.1  576.13   384.5 578.525     391  581.91
     395  582.97  427.61584.5596   438.9  589.14   450.9  596.42   506.7  620.84
#Mann= 7 ,-1 , 0
       0     .12       0   215.5    .045       0   243.4     .06       0
  280.15    .016       0  313.23     .12       0   384.5    .016       0
  427.61     .12       0
#XS Ineff= 2 , 0
                           281.9          579.49
Permanent Ineff=
       F       F
Bank Sta=215.5,243.4
XS Rating Curve= 0 ,0
Exp/Cntr=0.3,0.1

Type RM Length L Ch R = 1 ,16569.2 ,183.6,193.9,211.8
XS GIS Cut Line= 3
     2300188.228      398956.652     2300326.249      398896.756
     2300587.967      398657.173
#Sta/Elev= 30
       0  638.76    39.6  630.32    63.4  621.95    75.2  614.97    91.1  613.16
   102.9  606.04   138.6  589.05   166.4  572.53   170.4  571.55   182.4  572.81
     193  570.84   202.3  569.75     213  570.32  218.54571.0199   226.2  572.41
   246.1  572.49  257.55573.9844     286  574.58  300.93572.6295   305.9  571.71
   329.9  570.86   341.8  571.82   369.7  578.53  384.49583.1003   417.6  584.78
   421.6  585.52  429.93590.4505   461.4  598.24   485.3  607.07   505.3  616.16
#Mann= 8 ,-1 , 0
       0     .12       0     193    .045       0     213     .12       0
  218.54     .06       0  257.55    .016       0  300.93     .12       0
  384.49    .016       0  429.93     .12       0
#XS Ineff= 2 , 0
                          281.13          577.55
Permanent Ineff=
       F       F
Bank Sta=193,213
XS Rating Curve= 0 ,0
Exp/Cntr=0.3,0.1
